--- LtlKwhaRvr.prj (project) ---

Proj Title=LtlKwhaRvr
Current Plan=p01
Default Exp/Contr=0,0
English Units
Geom File=g01
Flow File=f01
Plan File=p01
BEGIN DESCRIPTION:
AMEC Environment & Infrastructure, 2013
Projection: NAD 1983 State Plane West Virginia South FIPS 4702 (US Feet)
Vertical Datum: NAVD 1988
END DESCRIPTION:
DSS Export Rating Curves= 0
DSS Export Rating Curve Sorted= 0
DSS Export Volume Flow Curves= 0
DXF OffsetX= 0
DXF OffsetY= 0
DXF ScaleX= 0
DXF ScaleY= 0

--- LtlKwhaRvr.p01 (plan) ---

Plan Title=Floodplain
Program Version=4.00
Geom File=g01
Flow File=f01
K Sum by GR=0
Std Step Tol=0.01
Critical Tol=0.01
Num of Std Step Trials=20
Max Error Tol=0.3
Flow Tol Ratio=0.001
Split Flow NTrial=30
Split Flow Tol=0.02
Split Flow Ratio=0.02
Log Output Level=0
Friction Slope Method=1
Unsteady Friction Slope Method=2
Unsteady Bridges Friction Slope Method=1
Global Log Level=0
CheckData=False
Run HTab=0
Run UNet=0
Run PostProcess=0
UNET Theta=0
UNET Theta Warmup=0
UNET ZTol=0
UNET ZSATol=0
UNET MxIter=0
UNET MaxInSteps=0
UNET DtIC=0
UNET DtMin=0
UNET MaxCRTS=0
UNET WFStab=0
UNET SFStab=0
UNET WFX=0
UNET SFX=0
UNET DSS MLevel=0
UNET DZMax Abort=0
UNET Convert EG Bridges=0
UNET Use Existing IB Tables=0
UNET Froude Limit=0
UNET Froude Power=0
Write IC File=0
Echo Input=False
Echo Output=False
Write Detailed=0

--- LtlKwhaRvr.f01 (steady flow) ---

Flow Title=NFF Regression Equation
Program Version=4.10
Number of Profiles= 1
Profile Names=P100yr
River Rch & RM=LtlKwhaRvr,Main            ,60521.3
20121.62
River Rch & RM=LtlKwhaRvr,Main            ,50576.4
   20203
River Rch & RM=LtlKwhaRvr,Main            ,50149.5
20669.05
River Rch & RM=LtlKwhaRvr,Main            ,30498.6
20920.65
River Rch & RM=LtlKwhaRvr,Main            ,29536.2
21526.05
River Rch & RM=LtlKwhaRvr,Main            ,16325.7
21863.86
River Rch & RM=LtlKwhaRvr,Main            ,15816.3
21935.06
River Rch & RM=LtlKwhaRvr,Main            ,717.8
22144.19
River Rch & RM=LtlKwhaRvr,Main            ,142.3
22149.89
Boundary for River Rch & Prof#=LtlKwhaRvr,Main            , 1
Up Type= 0
Dn Type= 3
Dn Slope=0.00068
DSS Import GetInterval= 0
DSS Import GetPeak= 0
DSS Import FillOption= 0

--- LtlKwhaRvr.g01 (geometry) ---

Geom Title=USGS 3m DEM
Program Version=4.10

River Reach=LtlKwhaRvr      ,Main
Reach XY= 30
     1905591.528      671414.576     1903468.197      672395.225
     1903437.797      674647.545     1902422.201      674510.063
     1900527.434      672750.629     1899599.933      674284.174
     1898370.275      674641.904     1898483.081      676826.786
     1899221.194      677373.903      1901015.31      676997.089
     1901414.737      677889.813      1901383.45      678546.318
      1899210.59      679308.224      1900777.42       680485.94
     1899455.472      682129.243     1900961.256      682525.292
     1899828.809      683995.643     1900674.581      685173.892
      1898974.23      685861.595     1894623.411      689232.535
     1894590.181       689654.28     1897691.705      690733.134
     1894388.791      692676.599     1894868.056       694746.89
     1893516.763       696061.59     1892144.766      694340.354
     1891377.104      694241.321     1891595.805      697153.952
     1889178.199      696598.059     1889605.528      697815.956

Type RM Length L Ch R = 1 ,60521.3 ,20.2,20.2,20.2
XS GIS Cut Line= 4
     1905283.068      670966.683      1905523.52      671286.995
     1905612.061      671519.634     1905738.798      672038.731
#Sta/Elev= 30
       0   792.5    39.1  804.06    48.8  805.32    58.6  804.68    68.4  802.18
     127  780.59   175.8   755.4   205.1   744.4   234.4   735.6   312.6  716.19
   361.4  707.07   371.2  703.61   390.8  693.16   400.5  689.37   438.8  682.25
   477.1  668.44   486.7  666.54   505.8   666.3   582.4  668.09   678.6  682.02
   727.2  686.55   756.3  693.44     766  698.14   775.7   704.7     834   747.7
     902  799.96   921.5  811.48  1057.5  868.74  1076.9  873.16  1183.8  887.19
#Mann= 3 , 0 , 0
       0      .1       0   477.1    .045       0   582.4      .1       0
Bank Sta=477.1,582.4
XS Rating Curve= 0 ,0
Exp/Cntr=0.3,0.1

Type RM Length L Ch R = 1 ,60501.1 ,62.6,62.5,62.5
XS GIS Cut Line= 4
     1905267.443      670982.308     1905507.895       671302.62
     1905596.436      671535.259     1905723.173      672054.356
#Sta/Elev= 30
       0  798.09    29.3  805.43    39.1  805.01    48.8  802.55   117.2   777.7
   166.1  752.32   205.1  738.12   312.6  712.91   429.2  689.42   448.4  683.36
   477.1  668.28   486.7  666.54   505.8   666.3   572.8  668.67   601.6  676.05
   639.9  683.37   678.6  686.68   707.7  686.98   736.9  691.49   746.6  695.08
   756.3  701.28   785.4  723.31     834  755.28   892.3  797.13   921.5  813.11
   999.2   845.7    1038  863.35  1057.5  870.01  1144.9  883.75  1183.8  888.44
#Mann= 3 , 0 , 0
       0      .1       0   477.1    .045       0   572.8      .1       0
Bank Sta=477.1,572.8
XS Rating Curve= 0 ,0
Exp/Cntr=0.3,0.1

Type RM Length L Ch R = 1 ,60438.5 ,262.3,261.7,261.1
XS GIS Cut Line= 4
     1905204.943      670992.724     1905445.395      671313.037
     1905533.936      671545.676     1905660.673      672064.773
#Sta/Elev= 30
       0  801.14    19.5  805.68    29.3  805.04    39.1  802.44   107.5   775.2
   156.3  753.01   195.4  736.95   214.9     732   312.6  713.05   351.7  703.06
   419.7  682.83   438.8  679.29   467.5  677.04   477.1   673.9   486.7  669.36
   496.3  666.85   515.4   666.3   563.3  666.91   582.4  668.21   611.1  674.79
   688.3  686.12   717.4  688.88   727.2  691.18   746.6  699.94   921.5  796.01
  1047.8  859.37  1076.9   869.2  1096.4  873.39  1144.9  880.67  1183.8  885.11
#Mann= 3 , 0 , 0
       0      .1       0   486.7    .045       0   582.4      .1       0
Bank Sta=486.7,582.4
XS Rating Curve= 0 ,0
Exp/Cntr=0.3,0.1

Type RM Length L Ch R = 1 ,60176.9 ,632.6,633.1,633.5
XS GIS Cut Line= 4
     1904808.242      671065.641     1905189.566      671378.394
     1905277.943      671594.766     1905515.707      672168.071
#Sta/Elev= 30
       0  869.35    19.3  866.58    38.7  858.75   106.4   818.9   193.4  775.05
   241.8   744.1   261.1   734.6   338.4   717.4   396.5  711.11   415.8  703.59
   454.5  683.72   464.2  680.74   502.9  677.35   551.6  676.98   561.4  675.54
   580.8  668.28   600.3  666.32   668.5  668.35   697.7  673.28   794.8  676.45
   833.6   685.3   862.7     690   911.2   716.2   969.3  753.25  1008.1  772.91
  1056.6  794.45  1134.2  823.03  1240.9  838.32  1289.4  841.91  1347.6  842.08
#Mann= 3 , 0 , 0
       0      .1       0   580.8    .045       0   668.5      .1       0
Bank Sta=580.8,668.5
XS Rating Curve= 0 ,0
Exp/Cntr=0.3,0.1

Type RM Length L Ch R = 1 ,59543.8 ,700.6,696.3,691.9
XS GIS Cut Line= 4
     1904383.763      671188.905     1904605.117      671592.551
     1904722.305       671900.71     1904982.721      672408.523
#Sta/Elev= 30
       0  883.57    58.8  878.66    88.2  871.78   107.7  865.58   127.3  856.65
   176.3   828.8   274.2  777.02     333  738.63   352.6  728.09   440.8  693.37
   479.8   679.9   499.1  675.58   528.2  674.67   557.3  666.91     567  665.92
   634.9  668.46     664  676.76   683.4  680.05   741.6  681.68   809.7  689.39
   858.9  691.98   868.8  695.74   888.4  707.16   908.1  716.18   986.8  744.02
  1085.2  786.62  1154.1  805.97  1193.5  823.61  1272.2  853.93  1360.7  882.23
#Mann= 3 , 0 , 0
       0      .1       0   557.3    .045       0   634.9      .1       0
Bank Sta=557.3,634.9
XS Rating Curve= 0 ,0
Exp/Cntr=0.3,0.1

Type RM Length L Ch R = 1 ,58847.5 ,785.3,771.7,758
XS GIS Cut Line= 4
     1903376.818      671214.946     1903945.395      671870.328
     1904123.346      672152.446     1904522.652      672721.023
#Sta/Elev= 30
       0  929.48   243.7  874.41   341.2  835.88     351  835.68   409.4  850.77
   487.4   852.3   516.7  847.39   653.2  787.63   682.4  768.65   721.4  738.41
   731.2  734.75   779.9  731.72   828.6  732.91   867.6  723.34   897.1  704.61
   946.1  667.01   955.9  665.05  1034.4  669.24  1063.8  677.69  1103.1  682.62
  1269.7  686.09    1299  689.22  1387.1  722.47  1465.4   759.2  1582.8  827.32
  1612.2  839.86  1719.8  851.26  1788.3  853.16  1837.3  849.75    1896  836.94
#Mann= 3 , 0 , 0
       0      .1       0   946.1    .045       0  1034.4      .1       0
Bank Sta=946.1,1034.4
XS Rating Curve= 0 ,0
Exp/Cntr=0.3,0.1

Type RM Length L Ch R = 1 ,58075.8 ,498.7,487.9,477.2
XS GIS Cut Line= 4
     1902678.034      672273.974     1903316.055      672417.203
      1903550.43       672517.03     1904418.485      672872.933
#Sta/Elev= 30
       0     885    68.3  885.86   136.6  882.14   224.5   872.7   302.6  857.06
   370.9  826.46   507.5  756.47   566.1  720.77   614.9   696.2   702.9   679.5
   732.3  669.78   761.7   663.8   820.5  664.56   830.3  668.83   849.9  676.26
  1016.2  687.72  1055.2  702.44  1094.3     722  1192.1     781  1250.7  796.95
    1280   799.1  1358.2  792.24  1455.9  760.36    1495  741.19  1534.1  734.68
  1563.4  742.08  1661.2     785  1719.8  802.72  1788.2  821.37  1846.8  827.48
#Mann= 3 , 0 , 0
       0      .1       0   732.3    .045       0   830.3      .1       0
Bank Sta=732.3,830.3
XS Rating Curve= 0 ,0
Exp/Cntr=0.3,0.1

Type RM Length L Ch R = 1 ,57587.9 ,818,817.2,816.1
XS GIS Cut Line= 4
     1902916.749      673003.141     1903303.034      672959.738
     1903580.811      672938.037     1904431.506      673111.648
#Sta/Elev= 30
       0  885.75    19.4  888.98   116.6  897.54     136  894.34   184.6  875.56
   204.1  862.63   252.7   824.7   301.2  780.97   340.1  741.06   359.6  723.74
     379  711.96   417.5  693.16   465.6  676.43   494.4  663.93   532.8  662.41
     552  663.52   619.3  671.69   764.9  678.33   833.2   688.6   950.2  686.56
     999  703.69  1067.3  713.35  1125.8  716.27  1262.4  727.73  1301.4  727.04
    1321  733.53  1369.7  761.18    1399  774.83  1447.8  789.12  1535.6  809.92
#Mann= 3 , 0 , 0
       0      .1       0   494.4    .045       0     552      .1       0
#XS Ineff= 2 , 0
                          832.11          694.73
Permanent Ineff=
       F       F
Bank Sta=494.4,552
XS Rating Curve= 0 ,0
Exp/Cntr=0.3,0.1

Type RM Length L Ch R = 1 ,56770.7 ,614.7,626.6,638.2
XS GIS Cut Line= 4
     1903099.041       673771.37     1903593.832      673684.565
     1903919.353      673645.502     1904635.499      673593.419
#Sta/Elev= 30
       0  805.88    38.6  797.24    96.6  801.18   154.6  800.34   173.9  798.06
   280.2   772.3   357.4   749.8   415.4  725.25     454  705.62     483  687.46
   492.7   683.8   540.9  671.76   627.7  672.05   637.4   671.1   656.6  664.27
   675.9   662.2   724.1   663.6   762.7  680.28   801.3  686.58   830.2  694.63
   889.2  719.88   958.1  735.02   997.4  736.64  1085.9  713.24  1115.4  710.92
  1154.8  721.92  1243.3  760.15  1282.7  770.02  1390.9  783.42  1548.2  786.02
#Mann= 3 , 0 , 0
       0      .1       0   656.6    .045       0   724.1      .1       0
Bank Sta=656.6,724.1
XS Rating Curve= 0 ,0
Exp/Cntr=0.3,0.1

Type RM Length L Ch R = 1 ,56144.1 ,620.6,643.8,667.1
XS GIS Cut Line= 4
     1903164.145      674036.127     1903580.811      674209.738
     1903845.568      674322.585     1904414.145      674626.405
#Sta/Elev= 30
       0  846.81    58.9  841.11   127.6  819.74   176.6  801.09     265  762.91
   343.4  725.36   441.6   690.5   537.7  677.11   576.1  670.04   585.7  666.16
   595.3  662.65   604.9  662.01   652.8  662.23   662.4  663.45     672  667.54
   681.6  672.36     720   686.7   739.2  698.34   836.9  770.06     915  833.52
   924.8  838.88   934.5  841.99   963.8  845.62  1081.1  853.87  1159.2  866.05
  1247.1  876.57  1286.2  882.72  1325.2  886.02  1354.6  884.43  1383.8  886.31
#Mann= 3 , 0 , 0
       0      .1       0   585.7    .045       0     672      .1       0
Bank Sta=585.7,672
XS Rating Curve= 0 ,0
Exp/Cntr=0.3,0.1

Type RM Length L Ch R = 1 ,55500.3 ,712.7,725.4,738.1
XS GIS Cut Line= 4
     1903020.916      674148.974     1903259.631      674457.134
     1903316.055       674856.44     1903350.777      675403.315
#Sta/Elev= 30
       0   846.7      39  845.28    87.7   838.3   116.9  830.39   253.4  765.88
   380.1     697   419.3  682.18   429.2  680.42   517.7  677.54     557  671.38
   576.7  663.72   596.4   661.8     675  662.44   694.7  664.91   734.1  679.74
   773.4   686.5   793.1  692.76   812.6  703.43     842  723.84   871.4  740.03
   910.5  765.93   939.9  777.19     979  797.86  1008.4  809.27  1057.3  831.54
  1155.1  863.76  1233.4  886.89    1253   889.6  1301.9   884.1    1341  873.67
#Mann= 3 , 0 , 0
       0     .07       0   576.7    .045       0   694.7      .1       0
Bank Sta=576.7,694.7
XS Rating Curve= 0 ,0
Exp/Cntr=0.3,0.1

Type RM Length L Ch R = 1 ,54774.9 ,516.4,530,543.6
XS GIS Cut Line= 4
     1902942.791      674122.933     1902647.652      674444.113
     1902513.103      674743.592     1902421.957      675273.106
#Sta/Elev= 30
       0  842.82    19.4   839.7    77.6  823.91   164.8  791.24   213.2  771.69
   300.5  724.37   416.8  680.96   455.5  673.28   532.8  670.47   561.7  662.58
     581   661.8   629.3   662.8   667.9  674.22     784  700.18   832.9  726.71
   891.5  770.17     911  778.81   930.6  784.17   950.1  780.05   979.4  766.99
  1028.3  731.37    1038  726.31  1086.9  715.03  1096.7  716.53  1106.4  722.44
    1126  738.72  1184.6  774.14  1262.7  818.16  1282.3  827.24  1301.8  833.51
#Mann= 3 , 0 , 0
       0     .07       0   561.7    .045       0   629.3      .1       0
Bank Sta=561.7,629.3
XS Rating Curve= 0 ,0
Exp/Cntr=0.3,0.1

Type RM Length L Ch R = 1 ,54244.9 ,484.6,482.6,480.6
XS GIS Cut Line= 4
     1902751.818      673858.176     1902326.471      674166.335
     1902057.374      674331.266     1901510.499      674782.655
#Sta/Elev= 30
       0  817.64    68.1  801.01   126.4   784.1   204.3  747.96   262.6  727.66
   291.8   718.8   379.3  698.49   496.1  677.47   515.5  675.13   620.9  670.23
   630.4  668.18     640   664.2   649.6  662.03   668.7   661.7     707  661.74
   726.1  664.22   745.2  671.02   754.8  672.72   821.7  680.79   986.6   683.9
  1015.7  688.74  1035.1  695.52  1112.8   740.8    1142   754.7  1239.1  783.36
  1316.8  813.21  1384.8  836.35  1404.3     840  1452.8  844.33    1550  848.56
#Mann= 3 , 0 , 0
       0     .06       0     640    .045       0   726.1     .06       0
Bank Sta=640,726.1
XS Rating Curve= 0 ,0
Exp/Cntr=0.3,0.1

Type RM Length L Ch R = 1 ,53762.3 ,885.6,880.6,875.5
XS GIS Cut Line= 4
     1902560.846      673337.342     1901979.249      673810.433
     1901697.131      674018.766     1901276.124      674374.669
#Sta/Elev= 30
       0   751.3    97.4  714.21   136.3  707.91     185  707.52   262.9  698.11
   408.9  693.68     516  686.16   593.9  691.22   681.6  682.38   749.7  683.26
   788.7  675.69   827.6  662.27   847.1   661.7   905.6  663.07   934.8  670.63
   973.8  670.49  1022.5  679.08  1139.1  681.22  1206.8  685.19  1235.8  692.29
  1264.8  703.67  1284.2  712.68  1313.2  729.74  1332.5  738.26  1409.9  751.24
  1458.3  767.29  1487.3  774.51  1516.3  779.71  1574.3  786.01  1651.7  804.85
#Mann= 3 , 0 , 0
       0     .06       0   827.6    .045       0   905.6     .06       0
#XS Ineff= 2 , 0
          716.39  693.33
Permanent Ineff=
       F       F
Bank Sta=827.6,905.6
XS Rating Curve= 0 ,0
Exp/Cntr=0.3,0.1

Type RM Length L Ch R = 1 ,52881.8 ,905.5,886.5,867.5
XS GIS Cut Line= 4
     1901660.673      672813.905     1901400.256      673100.363
     1901108.589      673438.905     1900978.381      674032.655
#Sta/Elev= 30
       0  843.35    96.8  820.36   154.8  798.16   164.5  796.22   193.6  797.67
   203.2  796.04   222.6  787.96   261.3  763.58   338.8  724.42   396.8  703.18
   455.1   683.8   503.7  671.47   523.1  664.06   542.6   661.7   591.1  661.71
   610.6  663.37   639.7  672.17   717.4  677.27   756.3  682.01   804.8   695.8
     834  701.52   892.8  701.94   951.6  716.66  1206.6  765.02  1255.6   768.1
  1265.4  771.19  1314.4  795.55  1343.8  807.85  1392.8  823.93  1441.8  836.92
#Mann= 3 , 0 , 0
       0      .1       0   523.1    .045       0   610.6     .07       0
Bank Sta=523.1,610.6
XS Rating Curve= 0 ,0
Exp/Cntr=0.3,0.1

Type RM Length L Ch R = 1 ,51995.3 ,789.1,775.8,762.5
XS GIS Cut Line= 4
     1900499.214      672089.946     1900535.673      672626.405
     1900587.756      673053.488     1900728.381      674100.363
#Sta/Elev= 30
       0  831.98    48.9  807.22   185.8  764.83   215.1  750.37   224.8  747.84
   283.5  755.75   361.7  775.07   410.6   778.1   430.2  775.88   449.7  767.71
   459.5  761.36   498.6  725.47     567  677.86   606.1  670.74   625.7  664.24
   645.3   661.7   723.5  663.13   752.8  671.52   840.8   686.5   860.4  688.06
   977.7  689.46  1104.9  694.73  1202.7  687.03  1280.9  694.86  1388.5  695.47
  1554.8  705.66  1652.6  719.22  1740.6  743.29  1848.2  768.78  2024.2  805.98
#Mann= 3 , 0 , 0
       0      .1       0   625.7    .045       0   723.5      .1       0
Bank Sta=625.7,723.5
XS Rating Curve= 0 ,0
Exp/Cntr=0.3,0.1

Type RM Length L Ch R = 1 ,51219.5 ,642.4,643.1,643.7
XS GIS Cut Line= 4
     1899728.381      672928.488     1900056.506      673246.196
     1900259.631      673464.946     1900436.714      674058.696
#Sta/Elev= 30
       0  878.07    77.7  888.39   145.8  893.99   165.2  892.17   213.8  878.32
   291.5  845.61   301.2  839.28   330.4  808.04   340.1  799.61   369.3  780.86
   417.9  744.88   495.2  697.07   524.1  674.74   533.8  668.67   543.4  664.62
     553  662.17   572.3  661.71   639.7  664.48   668.6  671.59     736  681.41
   794.6  683.83   883.1  684.22   902.8  686.38   981.4  700.67  1030.6  716.64
  1178.2  769.16  1227.3   784.3  1276.5  796.76  1296.2  800.46  1374.8  808.53
#Mann= 3 , 0 , 0
       0      .1       0   543.4    .045       0   639.7     .08       0
Bank Sta=543.4,639.7
XS Rating Curve= 0 ,0
Exp/Cntr=0.3,0.1

Type RM Length L Ch R = 1 ,50576.4 ,432.4,426.9,421.4
XS GIS Cut Line= 4
     1899316.923      672678.488     1899732.374      673739.165
     1899971.089      674034.304     1900491.923      674628.922
#Sta/Elev= 30
       0  849.89   117.8   869.6   176.8  866.21   392.8  810.13   412.4  813.16
   451.7  830.59   510.6  850.26   579.4  860.32   608.8  861.08   638.3  852.72
   726.7  808.38   805.2  782.45     874  747.92    1090  677.69  1119.5  674.18
  1236.5  677.42  1314.3  664.84  1362.8   661.3  1401.9  662.13  1411.7     665
  1450.6  676.96  1596.8  685.01  1645.6  696.55  1684.6  715.42  1762.7  764.62
    1792  778.57  1821.3   786.4  2065.2  820.03  2201.8     835  2309.2  840.13
#Mann= 3 , 0 , 0
       0     .08       0  1314.3    .045       0  1411.7     .07       0
Bank Sta=1314.3,1411.7
XS Rating Curve= 0 ,0
Exp/Cntr=0.3,0.1

Type RM Length L Ch R = 1 ,50149.5 ,1396.5,1396.1,1395.7
XS GIS Cut Line= 4
     1898082.548       674017.03     1899191.923      673933.696
     1899733.589      674345.155     1900072.131      675063.905
#Sta/Elev= 30
       0  873.34   107.4  865.65   292.8  820.54   439.1  807.92   546.5  764.42
   673.4  720.41   722.2  706.72     810  689.89   868.5  688.66  1112.5  699.08
  1355.4  676.44  1501.2   675.8  1540.1  669.62  1588.7  667.38  1608.1  661.92
  1656.7   660.4  1695.6  662.44  1724.7  674.18  1792.7  680.15  1890.8   682.8
  1910.4  686.82  1959.5  709.16  2037.9  761.83  2096.8  784.18  2322.4  809.93
  2410.7  806.71  2469.5  798.29  2489.1  790.45  2528.4  763.81  2587.2  735.27
#Mann= 3 , 0 , 0
       0     .07       0  1608.1    .045       0  1695.6     .07       0
Bank Sta=1608.1,1695.6
XS Rating Curve= 0 ,0
Exp/Cntr=0.3,0.1

Type RM Length L Ch R = 1 ,48753.4 ,942.2,925.4,908.5
XS GIS Cut Line= 4
      1897944.18      674364.165     1898230.638      674542.117
     1898486.714      674728.749     1899090.013      675158.436
#Sta/Elev= 30
       0  842.34    19.3  843.12    77.1  824.74   125.3   813.9   183.1  821.11
   221.6  823.38   240.9  823.97   260.2  820.92   289.1   802.9   337.2  768.27
   442.8  675.98   462.1  663.52   481.3  660.59   548.5  659.63   567.7  662.26
   606.1  670.51   625.3  679.68   634.9  682.33     810  682.93   858.8  684.61
   936.7  689.57  1034.2  704.32  1063.4  711.03  1180.4  751.66  1199.9  759.02
  1268.1  790.66  1307.1  804.08  1326.6  807.74    1346  807.63  1394.8  797.37
#Mann= 3 , 0 , 0
       0      .1       0   462.1    .045       0   567.7     .07       0
Bank Sta=462.1,567.7
XS Rating Curve= 0 ,0
Exp/Cntr=0.3,0.1

Type RM Length L Ch R = 1 ,47828   ,1021.3,1023.8,1022.7
XS GIS Cut Line= 4
     1897553.555      675605.485     1898221.957      675575.103
      1898569.18       675536.04      1899198.52      675631.526
#Sta/Elev= 30
       0  883.22   118.1  882.82   236.2   887.3   275.5   883.3   344.4  871.29
   423.1   840.8   531.3  779.28   619.9  748.27   688.5  704.31   727.3  682.26
   785.6  662.05   795.3  658.03   814.7     656   872.9  656.31   892.3  662.83
   911.7  671.42   940.9   678.6  1018.5   676.8  1087.1  689.25  1214.4  755.09
  1253.5  771.72  1273.1  776.84  1282.9  775.23  1312.3  763.66  1400.4  724.91
    1420  720.44  1429.8  723.64    1469  747.78  1498.4  760.84    1655   813.1
#Mann= 3 , 0 , 0
       0      .1       0   785.6    .045       0   892.3     .07       0
Bank Sta=785.6,892.3
XS Rating Curve= 0 ,0
Exp/Cntr=0.3,0.1

Type RM Length L Ch R = 1 ,46804.2 ,578.9,567.3,555.3
XS GIS Cut Line= 4
     1897727.166      676612.429     1898182.895      676595.068
     1898669.006      676556.006     1899432.895      676456.179
#Sta/Elev= 30
       0  837.05    58.2  850.64   174.7  873.89   194.1  875.16   213.5  871.73
   232.9  861.26   271.7  831.56   378.4  767.02   465.8  731.73   475.6  726.96
   504.8   708.4   573.1  683.81   621.9   660.4   631.6  656.76   641.4     656
   699.9  656.65   719.4   660.9   787.7  676.65   885.2  676.14   963.2  678.93
  1021.8  695.53  1070.5  706.97  1099.8  711.04  1138.8  712.49  1158.3  714.73
  1382.6  759.89  1450.8  770.76  1509.3  787.71  1694.6  861.64  1714.1  867.68
#Mann= 3 , 0 , 0
       0      .1       0   621.9    .045       0   719.4     .07       0
Bank Sta=621.9,719.4
XS Rating Curve= 0 ,0
Exp/Cntr=0.3,0.1

Type RM Length L Ch R = 1 ,46236.9 ,741.8,721.5,701.2
XS GIS Cut Line= 4
       1897644.7      677858.089     1898512.756      677150.624
      1898890.36      676890.207     1899432.895      676516.943
#Sta/Elev= 30
       0  881.88    49.1  872.21     108  839.24   137.5  819.09   235.8  792.46
   373.3  736.76   392.9   736.2     442  744.84   520.6  737.15   589.4  744.92
   638.5  757.33     776  767.96   805.5  761.44   844.8  742.99   893.9   727.5
   952.8  696.39   982.3  685.41  1041.2  679.89  1227.2   676.8  1305.3  658.97
  1334.5     656  1383.3  658.77  1510.2  703.57  1647.3  699.27  1814.4  733.45
    1952  772.64  2001.2  782.81  2089.6  817.58  2178.1  842.02  2237.1  862.83
#Mann= 3 , 0 , 0
       0     .08       0  1305.3    .045       0  1383.3     .06       0
Bank Sta=1305.3,1383.3
XS Rating Curve= 0 ,0
Exp/Cntr=0.3,0.1

Type RM Length L Ch R = 1 ,45515.5 ,488.3,486.7,485.2
XS GIS Cut Line= 4
     1899280.985      678057.742     1899289.666      677523.887
     1899311.367      677215.728     1899476.298      676538.644
#Sta/Elev= 30
       0  872.55   184.4  862.09   213.6  862.38   310.6  868.52   339.8  867.75
   368.9  862.17   417.4  839.24   446.6  821.03   504.8  771.03   543.6  743.73
   591.8   696.6   601.5  688.62   630.5  667.63   649.8   658.3   659.4  656.38
   678.7     656   707.7     656   717.4  656.92     727  660.23   746.3  666.25
   804.2  675.34  1029.3  678.99  1078.4  681.48  1147.1  692.81  1196.2  703.53
    1314   748.2  1343.4  760.92  1392.5  784.67    1471  829.97  1539.7  863.66
#Mann= 3 , 0 , 0
       0      .1       0   649.8    .045       0     727     .05       0
Bank Sta=649.8,727
XS Rating Curve= 0 ,0
Exp/Cntr=0.3,0.1

Type RM Length L Ch R = 1 ,45028.8 ,473.3,467.5,461.6
XS GIS Cut Line= 4
     1899836.541      677810.346     1899784.457      677480.485
     1899784.457      677220.068     1899780.117      676577.707
#Sta/Elev= 30
       0  826.49     9.8  831.06    39.3  840.52    49.1  842.89    58.9  843.33
    88.4  837.69   117.9  828.78   216.1  784.24   314.3  736.24   382.2  692.01
   420.8  669.29     440  659.49   449.7  656.78     469     656   507.6  656.02
   517.2  656.64   526.8  659.23   536.5  662.73   546.1  664.72   672.2  673.23
   711.2  677.31   837.7  678.56   896.1  686.73   925.3  692.83     974  701.01
  1012.9  717.42  1149.1  782.03  1158.9  787.82  1217.3  828.75  1236.7  838.76
#Mann= 3 , 0 , 0
       0      .1       0     440    .045       0   526.8     .05       0
Bank Sta=440,526.8
XS Rating Curve= 0 ,0
Exp/Cntr=0.3,0.1

Type RM Length L Ch R = 1 ,44561.3 ,753,771.8,790.6
XS GIS Cut Line= 4
     1900396.436       677714.86     1900270.568      677337.256
     1900196.784      677059.478     1900088.277       676473.54
#Sta/Elev= 30
       0  807.55    29.1  806.94    48.5  803.79    58.2  800.49    87.4  787.36
   145.6   765.6   242.7  733.61   349.5  693.67   426.8  674.67   484.2  665.69
   503.4  657.84   522.6     656   560.9  656.05   570.5  656.68   580.1  659.35
   599.2  664.55   675.9  674.71   861.3  677.02   880.8  679.48   910.1  688.59
   949.2  696.08     959  699.23   968.7  704.08  1007.8  726.54  1037.1  741.42
  1144.6  784.63  1164.1  795.58  1203.2  822.56    1252  849.76  1281.3  863.11
#Mann= 3 , 0 , 0
       0      .1       0   503.4    .045       0   580.1     .05       0
Bank Sta=503.4,580.1
XS Rating Curve= 0 ,0
Exp/Cntr=0.3,0.1

Type RM Length L Ch R = 1 ,43789.5 ,676.1,691,705.5
XS GIS Cut Line= 4
     1900583.068      677727.881     1900873.867      677133.262
     1901038.798      676872.846     1901273.173      676360.693
#Sta/Elev= 30
       0  810.45    38.9  816.97    58.4  813.76   233.6  754.64   272.6  746.86
   282.3  743.55     292   738.8   311.5  726.87     331   718.5   389.4  705.98
   447.8  697.03   632.7  675.12   758.2  666.03   767.9  663.98   777.5  659.95
   787.1  657.33   806.4     656   873.8   656.1   883.5  657.04   893.1  659.89
     922  672.23   960.5  692.15   999.3  708.86  1135.2  753.96  1242.1  795.07
  1261.5  805.47  1319.8  841.22  1368.3  866.27  1465.4  903.55  1533.4  932.26
#Mann= 3 , 0 , 0
       0      .1       0   777.5    .045       0   893.1      .1       0
Bank Sta=777.5,893.1
XS Rating Curve= 0 ,0
Exp/Cntr=0.3,0.1

Type RM Length L Ch R = 1 ,43098.5 ,477.7,481.8,485.8
XS GIS Cut Line= 4
     1900734.978      677779.964     1901164.666      677619.374
     1901490.186      677493.506     1901967.617      677384.999
#Sta/Elev= 30
       0  793.95    68.3  789.18    87.8  786.28   107.4  781.26   136.6  771.12
   185.4  751.93     205  741.76   234.2  724.32   253.8  714.87   331.8  688.63
   351.4  685.35   380.6  683.12   497.5  677.69   555.7  665.88     575  659.61
   584.8  656.78   604.1  655.92   652.6  656.34   662.3  657.29     672   660.1
   788.3  709.49   846.9   736.7   944.8  794.68     984  819.44  1032.9  852.16
  1042.7  857.19  1101.5  873.62    1170  897.09  1248.4  929.12  1297.3  954.58
#Mann= 3 , 0 , 0
       0      .1       0     575    .045       0     672      .1       0
Bank Sta=575,672
XS Rating Curve= 0 ,0
Exp/Cntr=0.3,0.1

Type RM Length L Ch R = 1 ,42616.7 ,450.7,469,487.3
XS GIS Cut Line= 4
     1900891.228      678144.547     1901251.471      678062.082
     1901568.311      678001.318     1902084.805      677957.915
#Sta/Elev= 30
       0  836.01    38.9   838.6    48.6  837.71    68.1  831.23   165.3  776.57
   204.2  750.71   243.1  727.42   272.3   712.4   330.7  686.68   350.1  682.43
   457.6  676.78   506.4  667.04     526  660.17   535.8  656.86   565.1   655.9
   623.7  656.28   633.5  657.19   643.3  661.87   672.6   687.7   682.4  692.53
   721.5  705.45   838.9  737.11   897.6   760.6     966  796.52   975.8  805.03
   995.3  826.25  1005.1  833.91  1014.9  839.35  1151.8  891.13  1210.5   907.9
#Mann= 3 , 0 , 0
       0      .1       0     526    .045       0   643.3      .1       0
Bank Sta=526,643.3
XS Rating Curve= 0 ,0
Exp/Cntr=0.3,0.1

Type RM Length L Ch R = 1 ,42147.7 ,674.7,695.5,716.3
XS GIS Cut Line= 4
     1900834.805      678200.971     1901247.131      678352.881
     1901585.673      678591.596     1901928.555      678860.693
#Sta/Elev= 30
       0  837.13    39.1  836.51    68.4  828.51   156.2  795.67   185.5  778.43
   195.3  774.59   253.9  760.59     293  747.83   371.1  714.28   439.4  688.16
   487.6  678.64   564.7  675.68   612.8  667.91   632.1  660.69   641.7  656.58
     661  655.93   709.2  657.12   728.4  663.65   786.2  691.36   834.4  710.31
   863.4   724.3   902.1  749.35   960.2  779.46     999  806.89    1028  833.21
  1057.1  847.49  1124.9  874.06  1192.7  897.23  1260.5  906.56  1289.5  904.07
#Mann= 3 , 0 , 0
       0      .1       0   632.1    .045       0   728.4     .08       0
Bank Sta=632.1,728.4
XS Rating Curve= 0 ,0
Exp/Cntr=0.3,0.1

Type RM Length L Ch R = 1 ,41452.2 ,446.5,443.9,441.4
XS GIS Cut Line= 4
     1900747.999      678248.714     1900821.784      678678.401
     1900834.805      678960.519     1900834.805      679090.728
#Sta/Elev= 30
       0  820.44    19.4  813.92    38.8  805.56   106.6  766.65     126  756.64
     281  691.38     310  684.26   329.4  680.97   348.8  679.02   445.7  679.71
   465.2  678.45   484.7  668.72   504.2   665.3   513.9  660.95   523.6  656.76
   543.1  655.72   591.8  656.03   601.5  656.82     621  661.08   650.2  668.93
     660   673.1   689.2  689.21   698.9  695.74   708.7  704.08   746.3  741.86
   755.6   748.9   764.9  753.29   820.7  769.38     830  768.82   848.6  763.31
#Mann= 3 , 0 , 0
       0      .1       0   513.9    .045       0     621     .08       0
#XS Ineff= 2 , 0
          454.85  684.61
Permanent Ineff=
       F       F
Bank Sta=513.9,621
XS Rating Curve= 0 ,0
Exp/Cntr=0.3,0.1

Type RM Length L Ch R = 1 ,41008.2 ,528.1,521.7,515.3
XS GIS Cut Line= 4
     1900166.402      677979.617     1900366.055      678717.464
     1900405.117       678973.54     1900465.881      679299.061
#Sta/Elev= 30
       0   791.6    58.8  764.28   166.6  730.63   186.2  719.25   215.6   697.8
   225.4  693.47   235.2     692   274.4  697.63     392  686.61   470.4  681.39
   617.4  679.04   656.6  677.15   812.4   679.2     822  677.33   841.1  669.04
   869.9  661.55   879.5  657.78   889.1  655.83   937.1   655.2   965.9  656.06
     985   662.1  1004.2  671.01  1042.9  693.99  1111.1  743.66  1159.8  775.07
  1257.2  820.23  1276.6  826.86  1315.6  833.55  1335.1  832.45  1354.6  825.28
#Mann= 3 , 0 , 0
       0      .1       0   869.9    .045       0     985      .1       0
#XS Ineff= 2 , 0
          793.65  684.31
Permanent Ineff=
       F       F
Bank Sta=869.9,985
XS Rating Curve= 0 ,0
Exp/Cntr=0.3,0.1

Type RM Length L Ch R = 1 ,40486.6 ,647.2,633,618.3
XS GIS Cut Line= 4
     1899649.909      678491.769      1899819.18       678812.95
     1899940.707      679082.047     1900379.075      679273.019
#Sta/Elev= 30
       0  839.93    19.6  831.37   107.9   788.2   127.6  776.62   176.6  745.06
   196.2  735.22   284.6  701.45   343.4  676.02   363.1  671.47   412.3  664.46
   422.1  661.26     432  657.28   441.8   655.3   510.7   655.1   530.4  655.75
   540.2  658.18   550.1  663.25   559.9  667.68   589.4  674.46   628.8  677.72
   638.6  678.93   648.5  681.32   707.1  705.82   775.4  731.67   843.7  750.32
   921.8  777.28   970.6  788.43  1019.4  801.19  1097.4  815.76  1136.5  821.86
#Mann= 3 , 0 , 0
       0      .1       0   422.1    .045       0   550.1     .08       0
Bank Sta=422.1,550.1
XS Rating Curve= 0 ,0
Exp/Cntr=0.3,0.1

Type RM Length L Ch R = 1 ,39853.5 ,384.1,371.7,359.3
XS GIS Cut Line= 4
     1898603.902       678652.36     1899111.714      679012.603
     1899545.742      679264.339     1900366.055      679333.783
#Sta/Elev= 30
       0  818.48    38.9  824.25    68.1  823.51     107  818.58   155.6  804.86
   184.8  793.93   243.2  766.86   379.4  696.67     428  676.35   447.5  677.61
   486.4  704.01     574   742.4   603.2  749.82   622.6  750.84     662  735.53
     721  704.38     780  663.48   789.9  656.81   809.5   653.6   868.6  655.26
   888.2  663.38     967  671.23  1104.7  676.33  1212.6  708.39  1330.2  728.49
  1516.4  742.73  1614.4  742.71  1653.6  745.85  1800.6  772.01  1947.6  801.68
#Mann= 3 , 0 , 0
       0      .1       0     780    .045       0   888.2     .06       0
#XS Ineff= 2 , 0
          615.38  750.29
Permanent Ineff=
       F       F
Bank Sta=780,888.2
XS Rating Curve= 0 ,0
Exp/Cntr=0.3,0.1

Type RM Length L Ch R = 1 ,39481.8 ,569.2,558.3,547.3
XS GIS Cut Line= 4
     1898395.568      679494.374     1899007.548      679472.672
     1899471.957      679459.651     1900426.818      679372.846
#Sta/Elev= 30
       0  825.77      68  851.03   136.1  863.01     243  854.38   427.7   868.5
   476.3  869.11   534.6  863.79   544.3  860.45     554   853.6   592.9  811.59
     622     785   680.1  745.95   786.6  657.76   796.3  653.86   805.9   653.1
     864  655.04   883.4  659.08   902.7  664.75   989.8   672.6  1067.3  677.95
    1165  680.75  1282.4  702.22  1448.7  722.06  1566.1  724.83  1634.6  721.14
  1693.3  726.01  1781.4  737.48  1918.4  774.75  1986.8  787.75  2035.8  792.53
#Mann= 3 , 0 , 0
       0      .1       0   786.6    .045       0   883.4     .05       0
Bank Sta=786.6,883.4
XS Rating Curve= 0 ,0
Exp/Cntr=0.3,0.1

Type RM Length L Ch R = 1 ,38923.5 ,903.5,893,882.5
XS GIS Cut Line= 4
     1898929.423      680279.964     1899419.874      679989.165
     1899701.992      679828.575     1900491.923      679368.506
#Sta/Elev= 30
       0  837.13    78.6  803.19   147.5  779.87   186.8  770.95   265.4  734.65
   304.8  721.47   324.4  726.79   393.2  763.56   432.6  775.01   442.4  774.82
   491.5  748.66   540.7  702.39   570.2  678.44   609.5   663.5   629.2   653.2
     639  652.75   698.1  655.44   717.7  660.79   796.4  678.15  1002.9  680.45
  1081.6     686  1150.4  695.24  1238.8  696.84  1297.8     703  1376.4  692.54
  1455.1  709.84  1592.7  727.56    1632  738.35  1730.3  774.44  1808.9  793.48
#Mann= 3 , 0 , 0
       0      .1       0   609.5    .045       0   717.7     .05       0
#XS Ineff= 2 , 0
                          796.61          679.42
Permanent Ineff=
       F       F
Bank Sta=609.5,717.7
XS Rating Curve= 0 ,0
Exp/Cntr=0.3,0.1

Type RM Length L Ch R = 1 ,38030.5 ,481.4,493.5,505.6
XS GIS Cut Line= 4
      1899511.02      680414.512     1900235.846      680423.193
     1900400.777      680167.117      1900600.43      679346.804
#Sta/Elev= 30
       0  782.01    68.6  772.02   146.9  755.28   176.3  754.88   235.1  759.61
   274.3  756.49   323.3  744.29   401.6  711.27     480  686.65   724.9  661.62
   734.7  655.55   744.5  652.31   754.4   651.8   823.1  653.83   842.8   659.4
   872.3  665.44    1000  671.93  1422.2     671  1441.8  671.69  1490.9  678.06
  1530.1     676  1569.4  676.89  1598.9  683.88  1647.9  704.02  1736.3   728.9
  1755.9  738.25  1795.2  761.94  1814.8  771.13  1834.5  777.21  1873.7  784.51
#Mann= 3 , 0 , 0
       0      .1       0   724.9    .045       0   842.8     .05       0
#XS Ineff= 2 , 0
                         1063.55          683.53
Permanent Ineff=
       F       F
Bank Sta=724.9,842.8
XS Rating Curve= 0 ,0
Exp/Cntr=0.3,0.1

Type RM Length L Ch R = 1 ,37537   ,458.3,477.9,497.6
XS GIS Cut Line= 4
     1899563.103       680527.36     1900583.068      680518.679
     1900824.388        680399.9     1901275.777      680113.442
#Sta/Elev= 30
       0  791.08    29.4  790.02   117.7  767.39   196.2  732.92   215.8  726.38
   225.6  726.32   294.2   741.3   372.7  754.48   470.8     750   666.9  723.46
   774.8   715.1   843.5   704.3   912.1  687.06   951.4   682.8  1029.6  678.46
  1096.8  660.94  1116.1   652.8  1135.3   651.8  1279.4  653.88    1289   654.4
  1308.4  659.62  1347.3  670.46  1434.8  677.35  1454.2  680.55  1493.1  689.81
  1590.3  718.47  1609.7   727.5  1668.1  763.89  1765.3   809.8  1823.6  848.52
#Mann= 3 , 0 , 0
       0      .1       0  1096.8    .045       0  1308.4     .08       0
Bank Sta=1096.8,1308.4
XS Rating Curve= 0 ,0
Exp/Cntr=0.3,0.1

Type RM Length L Ch R = 1 ,37059.2 ,534.7,532.8,530.2
XS GIS Cut Line= 5
     1898897.305      680495.386     1899656.853      680616.914
     1900416.402      680760.143     1900690.246      680885.119
     1901063.103      681055.282
#Sta/Elev= 30
       0   790.5    68.2  805.35    97.4  804.25   175.3  774.22   262.9  727.59
   360.3  692.83   379.7  694.08   457.6  717.98   642.6   760.6   710.8  769.31
   759.5   769.9     779  767.62   886.6   733.8   955.1  697.73   994.2  703.96
  1297.5  701.45  1444.3  679.64  1610.1  664.66  1629.5  657.57    1649   651.7
  1716.9  653.31  1746.1  659.63  1775.2  675.88  1940.7  805.71  1960.3  816.66
  2067.6  778.73  2077.4  778.29  2126.2  804.18  2204.2  831.33    2253  842.26
#Mann= 3 , 0 , 0
       0      .1       0  1629.5    .045       0  1746.1      .1       0
Bank Sta=1629.5,1746.1
XS Rating Curve= 0 ,0
Exp/Cntr=0.3,0.1

Type RM Length L Ch R = 1 ,36526.3 ,540.2,539.9,540
XS GIS Cut Line= 4
     1898365.186      681295.589     1899910.325      681095.936
     1900400.777      681291.249     1900656.853      681408.436
#Sta/Elev= 30
       0  881.63   137.2  859.51   215.6  831.21   284.2  798.57   313.6  802.56
   362.6  826.26   431.1  846.61   460.5  851.34   489.9  849.56   538.9  837.45
   607.5  800.73   734.9  749.52   793.7  730.93   891.7  706.79  1019.1  687.67
  1185.6  695.41    1264  685.43    1313  684.65    1460  693.72  1548.2  680.29
  1763.3  661.26  1792.6  650.87  1880.6  653.35  1900.2  660.85  1939.2  677.99
    2037  740.56  2134.4  791.44  2231.6  836.07    2251  835.38  2367.5  793.63
#Mann= 3 , 0 , 0
       0      .1       0  1763.3    .045       0  1900.2      .1       0
Bank Sta=1763.3,1900.2
XS Rating Curve= 0 ,0
Exp/Cntr=0.3,0.1

Type RM Length L Ch R = 1 ,35986.4 ,721.6,712,702.4
XS GIS Cut Line= 4
     1898786.193      681612.429     1899654.249      681529.964
     1899927.686       681625.45     1900413.798      681681.874
#Sta/Elev= 30
       0  877.33    39.2  874.86    88.2   864.7   127.4  848.43     196   808.9
   254.7  784.33   333.1  758.18   401.7  730.53   529.1  687.74   587.8  683.43
   685.8  670.47   910.6     670   958.8  659.73   978.2  651.76   997.5  650.56
  1084.4  653.09    1094  656.11  1103.7  662.28  1113.3  668.66  1151.9   685.2
  1200.7  713.29  1259.5  735.09  1298.6  754.84  1318.2  761.47  1337.8   761.6
  1406.3  748.06  1445.4  748.74  1504.2  761.23  1562.9  783.36    1651  806.26
#Mann= 3 , 0 , 0
       0      .1       0   958.8    .045       0  1103.7      .1       0
Bank Sta=958.8,1103.7
XS Rating Curve= 0 ,0
Exp/Cntr=0.3,0.1

Type RM Length L Ch R = 1 ,35274.4 ,461,434,407
XS GIS Cut Line= 4
     1899003.207      682016.075     1899276.645      682194.026
     1899701.992      682146.283     1900383.416       681786.04
#Sta/Elev= 30
       0  844.31    67.2  829.03   134.3  816.35   182.3  812.61   230.3   814.8
   249.5  808.96   278.3  796.97   316.6  778.04   326.2  771.23   355.4  737.66
   365.2  729.89     443  675.46   472.2  659.73   481.9  653.86   491.6  650.94
   501.3   650.5     550  652.03   569.4  656.63   588.9  661.45   637.5  668.08
   968.9  670.79   998.2  672.83  1056.7  683.54  1115.3  679.63  1193.3  683.35
  1212.8  687.15  1232.4  693.68  1339.7  736.04  1466.5  789.66    1525  803.08
#Mann= 3 , 0 , 0
       0      .1       0   472.2    .045       0   569.4     .06       0
Bank Sta=472.2,569.4
XS Rating Curve= 0 ,0
Exp/Cntr=0.3,0.1

Type RM Length L Ch R = 1 ,34840.4 ,992.1,1010.2,1028.2
XS GIS Cut Line= 4
     1898950.256      682791.393     1899766.228      682517.088
     1899859.978      682180.282     1900400.777      681833.783
#Sta/Elev= 30
       0  822.64    29.4  812.06    97.8  800.95   156.5  778.79   195.6  760.27
   205.4  758.62   273.9  766.01     362  764.63   430.4  748.18   479.3  733.32
   557.6  728.71   635.8  718.06   694.6  696.98   723.9  681.59   772.8  671.29
   802.2  669.36   860.8  670.17     958  653.72   996.8  655.34  1025.9   650.5
  1093.9  651.23  1113.3  656.47  1132.8  664.26  1152.2  666.12  1395.4   669.3
  1541.3  677.35  1658.1  718.15  1726.2  747.52  1813.8  789.33  1852.7  801.91
#Mann= 3 , 0 , 0
       0      .1       0   996.8    .045       0  1113.3     .06       0
Bank Sta=996.8,1113.3
XS Rating Curve= 0 ,0
Exp/Cntr=0.3,0.1

Type RM Length L Ch R = 1 ,33830.2 ,825.6,847.6,869.5
XS GIS Cut Line= 4
     1899966.749      682810.346     1900578.728      682441.422
      1900921.61      682241.769     1901420.742      681985.693
#Sta/Elev= 30
       0  788.94     186  791.39   283.9  780.11   362.2  762.53   420.9  745.86
   489.4   720.8   577.5  693.55   626.5   680.8   830.7  671.24   917.8  657.88
   937.2   650.8   946.8  650.52  1004.9  651.61  1014.6  653.62  1024.3  658.38
    1063  683.33  1170.4  776.53  1180.2  782.06  1190.1  784.44  1229.5  789.52
  1268.8  789.37  1308.2  786.63  1396.8  774.52  1436.1  764.99  1455.8   757.6
  1465.7  756.39  1524.7  780.15  1544.4  785.32  1593.6  791.23  1672.3  797.15
#Mann= 3 , 0 , 0
       0      .1       0   917.8    .045       0  1024.3      .1       0
Bank Sta=917.8,1024.3
XS Rating Curve= 0 ,0
Exp/Cntr=0.3,0.1

Type RM Length L Ch R = 1 ,32982.6 ,906.9,902.5,898.2
XS GIS Cut Line= 4
     1899858.242       682875.45     1900474.561      682866.769
     1900808.763      683049.061     1901277.513      683240.033
#Sta/Elev= 30
       0  787.38   117.4  774.86   234.8  755.84   293.5  750.04   322.9  745.82
   459.8  710.47   538.1  685.71   557.7  681.75     587   678.4     714  671.52
   782.3  661.51   792.1  658.68   811.6  650.91   821.4   650.7   889.7     651
   899.4  653.78   909.2  659.85   928.7  674.85   938.5   680.6   967.8  693.04
   977.5  698.71  1113.9  781.46  1152.8  803.14  1211.2  841.78  1259.9  870.99
    1328  908.66  1337.8  912.14  1357.2  915.78  1386.4  917.75  1503.2  912.69
#Mann= 3 , 0 , 0
       0      .1       0   792.1    .045       0   909.2      .1       0
Bank Sta=792.1,909.2
XS Rating Curve= 0 ,0
Exp/Cntr=0.3,0.1

Type RM Length L Ch R = 1 ,32080.1 ,689.7,672.9,656.1
XS GIS Cut Line= 4
      1899511.02      683417.985     1899788.798       683504.79
     1900179.423      683617.637     1900743.659      683526.492
#Sta/Elev= 30
       0  920.13    38.8   916.4   106.7  889.24   116.4  883.76   164.9     846
     194  815.41   213.4  797.78   261.9  770.92   300.7   740.6   310.4  734.25
   358.8  707.64   416.9  669.66   426.6   664.8   455.6  655.23   465.3  651.63
   484.6   650.7   552.4  651.26   571.8  657.89   581.4  660.89   620.2  667.92
     717  680.94   746.1  686.75   765.4   693.3   901.1  748.46   978.6  775.47
  1085.1  803.38  1104.5  805.74  1133.6  804.35    1182  805.81  1269.2  797.12
#Mann= 3 , 0 , 0
       0      .1       0   455.6    .045       0   571.8      .1       0
Bank Sta=455.6,571.8
XS Rating Curve= 0 ,0
Exp/Cntr=0.3,0.1

Type RM Length L Ch R = 1 ,31407.1 ,908.2,908.5,908.4
XS GIS Cut Line= 4
     1899232.374      684588.124     1899721.957      684270.415
     1900117.791      684072.499     1900685.499      683780.832
#Sta/Elev= 30
       0  798.69    68.1  794.34   233.4  777.84   262.6  778.35     321  784.49
   389.1  787.88   408.5  788.01     428   785.2   457.2  776.18   466.9  771.36
   476.6  764.47   544.7  700.72   564.2  686.02   573.9  680.33   593.5  673.32
   652.5   661.5   672.2  655.14     682  652.07   701.6   650.7   780.3  650.92
   809.8  655.61     859  662.19   947.5  667.75  1104.7   689.3  1173.5  700.82
  1222.6  711.52  1291.3  733.45  1487.7  775.99  1595.7  787.56  1664.4  787.52
#Mann= 3 , 0 , 0
       0      .1       0   672.2    .045       0   809.8     .06       0
Bank Sta=672.2,809.8
XS Rating Curve= 0 ,0
Exp/Cntr=0.3,0.1

Type RM Length L Ch R = 1 ,30498.6 ,520,539.4,559.3
XS GIS Cut Line= 4
     1899518.832       684723.54     1900425.082      684843.332
     1900784.457       684661.04     1902221.957      683905.832
#Sta/Elev= 30
       0  888.35      59  885.91   108.1  879.93   314.5  824.64   481.6  758.07
   530.8  743.18   579.9   733.9   619.2  722.82   717.6  688.33   815.8  667.18
   884.6  668.09   963.3   659.2   982.9  650.22  1002.6   648.4    1091     653
  1110.7   660.1    1386  663.05  1484.4  678.36    1632  710.88  1720.6  716.89
  1828.8  714.81  2133.9  688.78    2193  689.53  2350.4   679.1  2389.8   679.1
  2527.6  699.79  2675.2  746.88  2763.8  788.75  2842.5  816.42  2940.9  861.44
#Mann= 3 , 0 , 0
       0     .08       0   963.3    .045       0  1110.7      .1       0
Bank Sta=963.3,1110.7
XS Rating Curve= 0 ,0
Exp/Cntr=0.3,0.1

Type RM Length L Ch R = 1 ,29959.2 ,412,423,434.3
XS GIS Cut Line= 4
     1899430.291      684822.499     1900357.374       685129.79
     1900810.499      685322.499     1902419.874      685978.749
#Sta/Elev= 30
       0  869.43    68.4  858.46   273.5  792.62   410.2  737.05     459     731
   654.4   682.5     840  671.24  1063.6  671.18  1237.4  655.49  1266.3   648.4
  1333.9  658.18  1420.8  711.87  1547.6  805.68  1694.9  747.55  1871.7  690.72
  1891.3  689.39  1950.2  703.06  1989.5  690.22  2028.8  697.01  2077.9  691.82
  2156.4  708.46  2313.6  708.11  2480.5  730.75  2549.2  731.97  2608.1  724.35
  2676.9  735.75  2735.8  730.23  2883.1  763.19  3030.4  808.07  3207.1  843.01
#Mann= 3 , 0 , 0
       0     .08       0  1237.4    .045       0  1333.9      .1       0
Bank Sta=1237.4,1333.9
XS Rating Curve= 0 ,0
Exp/Cntr=0.3,0.1

Type RM Length L Ch R = 1 ,29536.2 ,549.3,558.5,565.9
XS GIS Cut Line= 4
     1899227.166      684905.832     1900169.874      685312.082
     1900440.707      685650.624     1900872.999      686244.374
#Sta/Elev= 30
       0  874.45    39.1  865.28    58.7  858.73   146.6  818.12     176  806.87
   283.5   782.2   361.7  754.02   430.2  733.49   498.6  708.37   645.2  673.82
   684.3  670.24  1199.9   667.4  1248.1  663.45  1267.4  659.55  1286.6   649.2
  1296.3  648.31  1344.4  651.83  1373.4  659.96  1392.6   667.3  1402.3  673.33
  1460.1  716.98  1518.8  764.47  1567.8  797.61  1714.7  860.05    1744  871.01
    1793  884.99  1851.8  895.87  1930.1  915.01  2008.4   921.5  2194.5   932.5
#Mann= 3 , 0 , 0
       0     .06       0  1267.4    .045       0  1373.4      .1       0
Bank Sta=1267.4,1373.4
XS Rating Curve= 0 ,0
Exp/Cntr=0.3,0.1

Type RM Length L Ch R = 1 ,28977.6 ,774.9,765.4,757.3
XS GIS Cut Line= 4
     1899149.041      684999.582     1899774.041       685442.29
     1899836.541      685707.915     1899930.291      686322.499
#Sta/Elev= 30
       0  856.85   147.3  796.16   176.8  785.52   235.7  777.13   314.2  736.72
   392.8  691.32   422.2  677.21   441.9  670.82   510.6  665.71   559.7  664.89
   677.5  665.36   814.6  668.28   873.1  664.45   882.9  661.35   892.6  655.44
   902.4  650.24   921.8  647.49  1009.6  649.23    1029   657.1  1067.9   668.1
  1077.6  672.24  1135.9  707.32  1223.4  763.66  1281.6  807.66  1339.9   848.7
  1359.4  859.28  1407.9  874.15  1456.5  882.55  1524.5  892.68  1660.5  908.52
#Mann= 3 , 0 , 0
       0     .07       0   892.6    .045       0    1029      .1       0
Bank Sta=892.6,1029
XS Rating Curve= 0 ,0
Exp/Cntr=0.3,0.1

Type RM Length L Ch R = 1 ,28212.2 ,865,862.5,859.7
XS GIS Cut Line= 4
     1898586.541      685296.457     1898862.582      685530.832
     1899164.666      685895.415     1899586.541      686541.249
#Sta/Elev= 30
       0   950.6    48.9  942.57   127.2   923.8   176.2  915.56   205.5  905.71
   254.5  880.16   332.8  828.79   371.8  809.77   555.4  698.04     652  664.66
   661.7  658.24   671.3  650.19     681  645.63   690.6  645.22     739  647.56
   758.3  653.13   777.6  659.08   825.9  664.98   933.2  667.42   982.1  670.73
    1109  702.49  1167.6  725.43  1206.6  733.59    1236  743.43  1314.1  781.15
  1372.6  805.09  1421.5  832.65  1480.1  853.52    1568  899.88    1607  914.81
#Mann= 3 , 0 , 0
       0      .1       0   661.7    .045       0   758.3     .07       0
Bank Sta=661.7,758.3
XS Rating Curve= 0 ,0
Exp/Cntr=0.3,0.1

Type RM Length L Ch R = 1 ,27349.7 ,465.1,466.7,468.2
XS GIS Cut Line= 4
     1898101.298      685556.874     1898326.992      686255.658
     1898700.256      686611.561     1899359.978      687175.797
#Sta/Elev= 30
       0  893.42    88.1  856.95   264.4  840.19   303.5  828.67   342.7   823.2
   401.4  806.21   479.8  774.16     607  735.59     656  715.35   685.4  713.88
   724.5  723.46   763.5  719.95     783  712.34   841.4  676.84     890  662.94
   909.5  653.56   919.2  647.51   938.7  645.23   997.1  648.24  1016.5  652.68
  1065.2  662.84  1162.5  662.35  1220.9  670.57  1376.9  674.87  1435.4  684.94
  1630.5   763.8    1689  781.16  1825.6  812.85  1952.4  829.02  2118.2  898.17
#Mann= 3 , 0 , 0
       0      .1       0   909.5    .045       0  1016.5      .1       0
Bank Sta=909.5,1016.5
XS Rating Curve= 0 ,0
Exp/Cntr=0.3,0.1

Type RM Length L Ch R = 1 ,26883   ,1103.5,1108.9,1114.2
XS GIS Cut Line= 4
     1896517.096       685871.11     1897938.971      686485.693
     1898329.596      686912.776     1898678.555      687548.193
#Sta/Elev= 30
       0  882.44    58.8   879.2   127.4  866.51   254.9  825.96   539.2  722.43
   637.2  696.92   764.7  689.36   774.5  691.23   803.9  712.69   852.9  731.09
     951   746.7  1058.8  751.52  1323.5  744.47  1558.8  767.09  1666.7  756.51
  1774.6  728.25  1853.1  674.26    1912  652.21  1931.6  645.22  1990.5  648.02
  2010.1  654.49  2059.1  665.35  2245.4  675.31  2333.5  702.12  2490.3  777.91
    2598  842.75  2656.8  887.19  2686.2  901.75  2764.6  910.42  2852.7  886.26
#Mann= 3 , 0 , 0
       0      .1       0    1912    .045       0  2010.1     .07       0
Bank Sta=1912,2010.1
XS Rating Curve= 0 ,0
Exp/Cntr=0.3,0.1
